--- BRUSHRN1.prj (project) ---

Proj Title=BRUSHRN1
Current Plan=p01
Default Exp/Contr=0,0
English Units
Geom File=g01
Flow File=f01
Plan File=p01
BEGIN DESCRIPTION:
Stream Name: Brushy Run (1)
Flood Zone: Approximate
Pendleton County, West Virginia
HEC-RAS Version: 5.0.7
Hydrology Method:
Regression equation/Gage weighting
END DESCRIPTION:
DSS Export Rating Curves= 0
DSS Export Rating Curve Sorted= 0
DSS Export Volume Flow Curves= 0
DXF OffsetX= 0
DXF OffsetY= 0
DXF ScaleX= 0
DXF ScaleY= 0

--- BRUSHRN1.p01 (plan) ---

Plan Title=Floodplain
Program Version=5.07
Short Identifier=Floodplain
Geom File=g01
Flow File=f01
Subcritical Flow
K Sum by GR= 0
Std Step Tol= 0.01
Critical Tol= 0.01
Num of Std Step Trials= 20
Max Error Tol= 0.3
Flow Tol Ratio= 0.001
Split Flow NTrial= 30
Split Flow Tol= 0.02
Split Flow Ratio= 0.02
Log Output Level= 0
Friction Slope Method= 1
Unsteady Friction Slope Method= 2
Unsteady Bridges Friction Slope Method= 1
Parabolic Critical Depth
Global Vel Dist= 0 , 0 , 0
Global Log Level= 0
CheckData=True
Encroach Param=-1 ,0,0, 0
Mapping Interval=1HOUR
Computation Time Step Use Courant=        0
Computation Time Step Use Time Series=    0
Computation Time Step Count To Double=0
Computation Time Step Max Doubling=0
Computation Time Step Max Halving=0
Computation Time Step Residence Courant=0
Run HTab= 0
Run UNet= 0
Run Sediment= 0
Run PostProcess= 0
Run WQNet= 0
Run RASMapper= 0
UNET Theta= 0
UNET Theta Warmup= 0
UNET ZTol= 0
UNET ZSATol= 0
UNET MxIter= 0
UNET Max Iter WO Improvement= 0
UNET MaxInSteps= 0
UNET DtIC= 0
UNET DtMin= 0
UNET MaxCRTS= 0
UNET WFStab= 0
UNET SFStab= 0
UNET WFX= 1
UNET SFX= 1
UNET 1D Methodology=Finite Difference
UNET DSS MLevel= 1
UNET Pardiso=0
UNET DZMax Abort= 0
UNET Use Existing IB Tables= 0
UNET Froude Reduction=False
UNET Froude Limit= 0
UNET Froude Power= 0
UNET D1 Cores= 0
UNET D2 Coriolis=0
UNET D2 Cores= 0
UNET D2 Theta= 1
UNET D2 Theta Warmup= 1
UNET D2 Z Tol= 0.01
UNET D2 Volume Tol= 0.01
UNET D2 Max Iterations= 20
UNET D2 Equation= 0
UNET D2 RampUpFraction=0.1
UNET D2 TimeSlices= 1
UNET D2 BCVolumeCheck=0
UNET D1D2 MaxIter= 0
UNET D1D2 ZTol=0.01
UNET D1D2 QTol=0.1
UNET D1D2 MinQTol=1
Write IC File= 0
Write IC File at Fixed DateTime=0
Write IC File at Sim End=0
Echo Input=False
Echo Parameters=False
Echo Output=False
Write Detailed= 0
HDF Write Warmup=0
HDF Write Time Slices=0
HDF Flush=0
HDF Face Node Velocities=0
HDF Compression= 1
HDF Chunk Size= 1
HDF Spatial Parts= 1
HDF Use Max Rows=0
HDF Fixed Rows= 1
Calibration Method= 0
Calibration Iterations= 20
Calibration Max Change=0.05
Calibration Tolerance=0.2
Calibration Maximum=1.5
Calibration Minimum=0.5
Calibration Optimization Method= 1
WQ AD Non Conservative
WQ ULTIMATE=-1
WQ Max Comp Step=1HOUR
WQ Output Interval=15MIN
WQ Output Selected Increments= 0
WQ Output face flow=0
WQ Output face velocity=0
WQ Output face area=0
WQ Output face dispersion=0
WQ Output cell volume=0
WQ Output cell surface area=0
WQ Output cell continuity=0
WQ Output cumulative cell continuity=0
WQ Output face conc=0
WQ Output face dconc_dx=0
WQ Output face courant=0
WQ Output face peclet=0
WQ Output face adv mass=0
WQ Output face disp mass=0
WQ Output cell mass=0
WQ Output cell source sink temp=0
WQ Output nsm pathways=0
WQ Output nsm derived pathways=0
WQ Output MaxMinRange=-1
WQ Daily Max Min Mean=-1
WQ Daily Range=0
WQ Daily Time=0
WQ Create Restart=0
WQ Fixed Restart=0
WQ System Summary=0
WQ Write To DSS=0
WQ Use Fixed Temperature=0
Sorting and Armoring Iterations= 10
XS Update Threshold= 0.02
Bed Roughness Predictor= 0
Hydraulics Update Threshold= 0.02
Energy Slope Method= 1
Volume Change Method= 1
Sediment Retention Method= 0
XS Weighting Method= 0
Number of US Weighted Cross Sections= 1
Number of DS Weighted Cross Sections= 1
Upstream XS Weight=0
Main XS Weight=1
Downstream XS Weight=0
Number of DS XS's Weighted with US Boundary= 1
Upstream Boundary Weight= 1
Weight of XSs Associated with US Boundary= 0
Number of US XS's Weighted with DS Boundary= 1
Downstream Boundary Weight= 0.5
Weight of XSs Associated with DS Boundary= 0.5
Percentile Method= 0
Sediment Output Level= 3
Mass or Volume Output= 0
Output Increment Type= 1
Profile and TS Output Increment= 1
XS Output Flag= 0
XS Output Increment= 10
Write Gradation File= 0
Read Gradation Hotstart= 0
Write HDF5 File= 1
Write Binary Output= 1
Write DSS Sediment File= 0
SV Curve= 0
Specific Gage Flag= 0

--- BRUSHRN1.f01 (steady flow) ---

Flow Title=Flows
Program Version=5.07
Number of Profiles= 6
Profile Names=P100yr,P10yr,P25yr,P50yr,P500yr,P101yr
River Rch & RM=BRUSHRN1,Main            ,16811
     909     393     580     739    1377    1199
River Rch & RM=BRUSHRN1,Main            ,14990
    1022     445     654     832    1545    1335
River Rch & RM=BRUSHRN1,Main            ,11411
    1154     506     740     940    1741    1494
River Rch & RM=BRUSHRN1,Main            ,9911
    1503     666     968    1227    2261    1915
River Rch & RM=BRUSHRN1,Main            ,8111
    1671     743    1078    1365    2511    2117
River Rch & RM=BRUSHRN1,Main            ,0
    2918    1311    1890    2388    4378    3618
Boundary for River Rch & Prof#=BRUSHRN1,Main            , 1
Up Type= 0
Dn Type= 1
Dn Known WS=1259.25
Boundary for River Rch & Prof#=BRUSHRN1,Main            , 2
Up Type= 0
Dn Type= 1
Dn Known WS=1257.33
Boundary for River Rch & Prof#=BRUSHRN1,Main            , 3
Up Type= 0
Dn Type= 1
Dn Known WS=1258.21
Boundary for River Rch & Prof#=BRUSHRN1,Main            , 4
Up Type= 0
Dn Type= 1
Dn Known WS=1258.93
Boundary for River Rch & Prof#=BRUSHRN1,Main            , 5
Up Type= 0
Dn Type= 1
Dn Known WS=1259.95
Boundary for River Rch & Prof#=BRUSHRN1,Main            , 6
Up Type= 0
Dn Type= 1
Dn Known WS=1259.61
DSS Import GetInterval= 0
DSS Import GetPeak= 0
DSS Import FillOption= 0

--- BRUSHRN1.g01 (geometry) ---

Geom Title=Geometry
Program Version=5.07

River Reach=BRUSHRN1        ,Main
Reach XY= 30
2476848.55062059662261.7218946672476594.74497128662413.371105596
2476498.65440702662618.0713877832476629.78628778662885.445087388
2476367.12264869663606.6369139852475641.14744493664191.469798222
2474864.38653517665156.2337095592474382.24823493665984.388736576
 2474073.9461605666202.4234226352473956.35659611666720.528812274
 2473665.6348469666992.921047553 2473733.0461317667708.637826815
 2473627.2057839668273.7792951022472458.19306296668911.881932333
2471421.57171986669162.2686755512471061.82838938669613.464598089
2471206.71957353 669928.383524092471045.63951644670116.078824699
2470721.52694067 670240.084156932470067.10464311670289.730036899
2469638.30136651670669.2637994292469492.03713667670917.953638747
2469169.06174022672020.407388732 2469097.2259168672587.543396324
2468846.49516588672658.100866556 2468609.8647947672963.749386102
2468412.17987999673272.7311839012468402.15937576673540.297440737
2467904.24049556 673565.420420172467858.90970787673763.631603837

Type RM Length L Ch R = 1 ,16811   ,174.8,194.2,205.6
XS GIS Cut Line= 3
2476476.16605524662038.014012245     2476843.698      662270.466
2477104.63920453662419.735257687
#Sta/Elev= 30
       0 1476.05    26.7 1467.82    50.4 1463.16   112.7 1456.76   130.8 1453.75
   149.8 1451.76   182.9 1450.75   192.4 1448.85   196.8 1448.97   202.6  1450.7
   263.6 1449.41   338.8  1453.1   375.8 1453.92   396.8 1453.12   417.6  1450.3
   433.7 1448.78   443.8 1450.15   456.8 1451.69   539.8 1453.59   548.5 1454.74
   595.1 1467.04   636.5  1473.7   659.6 1478.59   666.1 1480.67   677.4 1485.87
   683.7 1487.55   710.3 1487.37   715.9 1489.45   727.6 1495.47   735.5 1498.46
#Mann= 9 ,-1 , 0
       0      .1       0  146.06     .05       0  278.71      .1       0
  314.57     .05       0  411.35      .1       0   417.6    .045       0
   443.8      .1       0  539.98     .05       0   620.7     .06       0
#XS Ineff= 2 , 0
           376.9 1457.65
Permanent Ineff=
       F       F
Bank Sta=417.6,443.8
XS Rating Curve= 0 ,0
Exp/Cntr=0.3,0.1

Type RM Length L Ch R = 1 ,16617   ,427.9,407.2,390.7
XS GIS Cut Line= 4
2476383.13252637662093.5147975512476684.29637763662254.985090107
2476708.59190802662430.467205139 2476990.7769773 662523.98830112
#Sta/Elev= 30
       0 1509.14    33.2 1495.93    58.6 1487.99    99.4 1477.06   108.5 1475.54
   126.6 1470.71   163.8 1465.27     246 1450.16   271.9 1448.03   281.4 1449.81
     340 1447.84   410.3 1448.72   465.3 1447.73   482.1 1444.95   487.4 1447.45
   495.1 1452.13   503.2 1453.83   518.9 1452.21   590.5 1451.97   647.5 1466.77
   672.8 1471.35   701.3 1474.34     714 1477.21   723.7  1481.1   731.8 1481.64
     752 1480.29   758.3 1482.69   769.8 1491.24   774.1 1493.44   816.2 1508.48
#Mann= 8 ,-1 , 0
       0      .1       0  264.46     .05       0  276.31      .1       0
   465.3    .045       0   487.4      .1       0  497.43      .1       0
  678.31      .1       0  685.55     .06       0
Bank Sta=465.3,487.4
XS Rating Curve= 0 ,0
Exp/Cntr=0.3,0.1

Type RM Length L Ch R = 1 ,16209   ,323.3,325.6,319.8
XS GIS Cut Line= 2
2476242.64340899662642.4831843542476890.94809698662737.490520245
#Sta/Elev= 30
       0 1496.05    16.3 1495.48    32.2 1493.22      58 1493.36      89 1489.17
   121.4 1483.72   145.6 1478.12   194.4 1457.59   226.5 1449.66   247.3 1440.85
   254.8 1438.47   262.9 1439.19     271 1440.86   295.2 1441.08   307.3 1443.25
   335.6 1444.46   404.4 1445.18   448.8 1444.65     465 1446.41   529.7 1463.76
   537.8  1467.2   550.5 1475.26     554 1476.19   570.1 1475.14   574.2 1475.45
   578.2 1477.66   590.3 1489.51   594.4 1492.05   622.7 1504.43   655.2 1516.48
#Mann= 4 ,-1 , 0
       0      .1       0   247.3    .045       0     271     .05       0
  457.91     .06       0
#XS Ineff= 2 , 0
                          346.62         1454.22
Permanent Ineff=
       F       F
Bank Sta=247.3,271
XS Rating Curve= 0 ,0
Exp/Cntr=0.3,0.1

Type RM Length L Ch R = 1 ,15884   ,260.4,262.8,265.3
XS GIS Cut Line= 2
2476196.01488465662868.953623347      2477012.51      663016.883
#Sta/Elev= 30
       0 1496.19    15.9 1494.96    51.6 1483.62    59.7 1478.86    71.9 1478.77
   116.6 1468.57   145.1 1467.43   181.6 1454.11   230.4 1449.43   250.7 1441.94
     300 1442.55     331 1441.07   356.4 1436.62   405.2 1439.16   413.6 1436.77
   421.5 1434.42   437.7 1437.33   437.7 1437.37   451.4 1443.68   466.2 1447.86
   526.9 1457.34   571.9 1461.37     580 1463.87   592.2 1470.56   612.5 1470.86
   624.7  1467.8   639.1 1467.26   661.6 1467.98   710.1 1472.75   829.8 1510.54
#Mann= 8 ,-1 , 0
       0     .05       0  234.34    .055       0  339.68    .035       0
  341.15     .05       0   413.6    .045       0   437.7     .05       0
  550.37     .06       0  655.71      .1       0
#XS Ineff= 2 , 0
          405.46  1442.6
Permanent Ineff=
       F       F
Bank Sta=413.6,437.7
XS Rating Curve= 0 ,0
Exp/Cntr=0.3,0.1

Type RM Length L Ch R = 1 ,15621   ,313.5,313,310.3
XS GIS Cut Line= 2
2476221.50283637663090.707715737     2476925.489      663324.341
#Sta/Elev= 30
       0 1492.89      26 1493.01    42.3 1491.67    51.9 1486.99    68.7 1474.21
    77.2 1469.32     132 1448.38     153 1439.07   157.2 1438.29   174.1 1439.76
   220.5 1438.76   233.1 1435.23   247.9    1436     309 1434.92   317.1 1432.39
     330  1430.5   334.3 1430.77   338.5 1432.77     346 1436.52   355.3 1438.02
   401.7 1438.74   431.2 1437.63   456.8 1448.97   513.8 1461.66     545  1471.5
   557.6 1478.32   578.7 1480.29     596 1492.83   673.6 1528.53   741.7 1556.45
#Mann= 10 ,-1 , 0
       0      .1       0   36.81     .05       0  148.84    .055       0
  183.08    .035       0  260.88     .05       0   317.1    .045       0
   338.5     .05       0  484.95    .055       0  596.98     .06       0
  610.04      .1       0
#XS Ineff= 2 , 0
          283.81 1440.48
Permanent Ineff=
       F       F
Bank Sta=317.1,338.5
XS Rating Curve= 0 ,0
Exp/Cntr=0.3,0.1

Type RM Length L Ch R = 1 ,15308   ,99.7,96.6,93.6
XS GIS Cut Line= 3
2476122.39809406663302.2496870752476287.33871991663454.661065397
2476716.76004299663547.775648254
#Sta/Elev= 30
       0 1492.05    33.1 1491.94    49.5 1490.58    57.3 1487.19    82.8 1472.53
   109.4 1463.77   180.2 1450.41     202 1444.94   234.4 1433.04   273.1 1432.92
   289.5 1430.85   330.4 1430.45   348.7 1428.82   354.9 1426.39   368.9  1428.7
   385.7 1435.83   391.8 1437.32     445 1438.33   477.7 1436.82   498.2  1444.1
   555.5 1455.27   563.7 1458.33   571.9 1463.06   577.4 1463.88   596.4 1463.31
   604.4 1467.42   617.8 1479.69   624.5 1484.03   640.9 1490.93     664 1498.81
#Mann= 6 ,-1 , 0
       0      .1       0  105.44     .05       0  252.38     .06       0
   348.7    .045       0   368.9    .055       0  572.49     .06       0
#XS Ineff= 2 , 0
          298.49 1435.75
Permanent Ineff=
       F       F
Bank Sta=348.7,368.9
XS Rating Curve= 0 ,0
Exp/Cntr=0.5,0.3

Type RM Length L Ch R = 1 ,15211   ,44,46,43
XS GIS Cut Line= 3
2476116.49356644 663333.089566442476354.17833645663572.945070828
2476701.89260904663578.009728519
#Sta/Elev= 30
       0 1491.99    22.7 1491.89    45.3 1490.39    77.1 1473.03    99.8 1466.18
   107.5 1462.77   205.3 1445.14   220.7 1440.14   237.6 1433.14   271.6  1432.6
   287.3 1430.24   306.6 1429.53   334.8 1430.02   358.2 1427.94   366.2 1425.45
   378.2 1427.65   382.2 1429.06   409.3 1430.66   438.3 1434.46   470.2 1436.22
   501.8 1436.55   517.6 1443.01   550.3 1447.79   574.3 1453.15   590.3 1459.07
   622.3 1459.31   630.3 1464.43   642.3 1477.19   646.3 1480.06   685.4 1493.94
#Mann= 9 ,-1 , 0
       0      .1       0  130.36     .05       0  301.25     .06       0
  309.17    .055       0   358.2    .045       0   378.2    .055       0
  417.04     .05       0   517.9    .055       0  618.76     .06       0
#XS Ineff= 2 , 0
          336.79    1427  391.48            1427
Permanent Ineff=
       F       F
Bank Sta=358.2,378.2
XS Rating Curve= 0 ,0
Exp/Cntr=0.5,0.3

Type RM Length L Ch R = 1 ,15165   ,9.2,18.3,35.2
XS GIS Cut Line= 3
2476091.89524832663343.7663878112476348.32741395663612.654525509
 2476677.4952601663612.654525509
#Sta/Elev= 30
       0 1490.98     9.9 1491.91    38.9 1491.98    66.5 1489.52    97.6  1473.2
   120.2 1465.81   131.5 1461.16   213.6 1446.91   247.5 1438.35   267.3 1434.47
   288.1 1431.46   308.3 1429.79   346.6 1427.99   363.6 1428.19   371.81426.607
     382 1424.68     394 1425.12   399.7 1426.76     410 1429.34     522 1435.32
     530  1437.3     538 1441.17     578 1446.05     614 1455.09     630 1455.95
     650 1455.01     658  1458.6   668.2 1465.74     678 1470.68   700.7 1476.69
#Mann= 9 ,-1 , 0
       0      .1       0  177.94     .05       0  296.74    .055       0
   371.8    .045       0   399.7    .055       0  463.02     .05       0
  563.63    .055       0  606.88     .06       0  664.24      .1       0
#XS Ineff= 2 , 0
          312.66 1432.88  422.94         1433.04
Permanent Ineff=
       F       F
Bank Sta=371.8,399.7
XS Rating Curve= 0 ,0
Exp/Cntr(USF)=0,0
Exp/Cntr=0.5,0.3

Type RM Length L Ch R = 1 ,15147   ,9.7,27.7,46.6
XS GIS Cut Line= 2
2476083.57715652663347.851354009 2476590.9172589663880.960608438
#Sta/Elev= 30
       0 1493.38     4.4 1491.06     7.2 1490.67    18.5 1492.19    45.2 1492.04
    72.3 1489.69      80 1486.41   100.6 1474.26     138 1460.76   219.3 1446.53
   236.4 1441.91   270.3 1434.87   300.5 1430.43   346.5 1427.84   364.3 1428.23
   373.91426.313   379.7 1425.05   385.2 1425.64   462.7 1430.77   484.6 1430.71
   503.6 1432.08   530.6 1432.55     608  1435.8   633.7 1439.03   661.3 1445.93
   688.9 1448.61   708.9 1448.05   716.5 1451.45   727.6 1458.89   735.9 1462.49
#Mann= 8 ,-1 , 0
       0      .1       0  174.45     .05       0  293.17    .055       0
   373.9    .045       0   385.2    .055       0  411.88     .05       0
   530.6    .055       0  547.74     .06       0
#XS Ineff= 2 , 0
          317.81 1432.68  441.55         1432.25
Permanent Ineff=
       F       F
Bank Sta=373.9,385.2
XS Rating Curve= 0 ,0
Exp/Cntr(USF)=0,0
Exp/Cntr=0.5,0.3

Type RM Length L Ch R = 1 ,15119   ,66.6,60.6,58.2
XS GIS Cut Line= 4
2476082.34410013663359.6856629272476333.15585346663615.596128558
 2476305.8684945663710.7218951642476581.32521177663899.812989263
#Sta/Elev= 30
       0 1490.62    15.7 1492.05    38.1 1492.02    66.1 1489.73    71.7 1487.33
    88.5    1477     132 1460.67   200.5 1448.79   231.7 1441.18   282.6 1431.56
   336.3 1427.76   365.4 1427.78   377.1 1425.94   386.7 1424.31   400.5 1425.84
   428.3 1428.61   453.5 1429.78   584.8 1432.62   607.6  1434.3   627.2 1437.69
   655.5 1440.42   669.6 1446.92   683.8 1452.03   690.8 1453.41     705 1453.98
   740.3 1451.25   747.4 1454.38   757.2 1464.05   760.1 1466.01   791.4 1473.06
#Mann= 7 ,-1 , 0
       0      .1       0  162.12     .05       0  282.07    .055       0
   377.1    .045       0   400.5    .035       0  520.37    .055       0
  661.76     .06       0
#XS Ineff= 2 , 0
          363.13    1427  418.61            1427
Permanent Ineff=
       F       F
Bank Sta=377.1,400.5
XS Rating Curve= 0 ,0
Exp/Cntr=0.5,0.3

Type RM Length L Ch R = 1 ,15059   ,79.4,68.4,53.2
XS GIS Cut Line= 4
2476058.74850128663379.5600848242476285.42976377663599.212268396
2476252.35597462 663726.878502172476534.32978794663947.616404066
#Sta/Elev= 30
       0 1494.24       8 1489.18    13.7 1487.71    22.2 1488.46    27.8 1491.28
    72.4 1488.93    79.5 1486.95    89.1 1480.23    98.5 1476.19   146.6  1458.5
   194.7 1451.66     229 1442.12     252 1438.33   268.3 1433.38   297.9 1429.69
   348.4 1428.16   372.31424.848   381.4 1422.23   393.8 1425.01   402.1 1427.99
   473.5  1427.6   543.3 1430.05   577.6 1433.04   617.3 1433.01   651.5 1442.39
   694.3 1460.17   728.5 1459.75   733.1 1462.02   750.3 1475.31   805.6 1488.24
#Mann= 12 ,-1 , 0
       0      .1       0    22.9     .05       0   68.41      .1       0
  145.15     .05       0   267.4    .055       0   372.3    .045       0
   393.8    .035       0  435.94     .05       0   454.4    .035       0
  496.17    .055       0  629.79     .06       0  763.41      .1       0
#XS Ineff= 2 , 0
          349.41 1433.66  420.49         1433.29
Permanent Ineff=
       F       F
Bank Sta=372.3,393.8
XS Rating Curve= 0 ,0
Exp/Cntr(USF)=0,0
Exp/Cntr=0.5,0.3

Type RM Length L Ch R = 1 ,14990   ,306.2,299.6,292.2
XS GIS Cut Line= 2
2476016.56532254663401.6573876832476438.13517328664037.406294436
#Sta/Elev= 30
       0 1496.36     2.5 1492.33     6.3 1489.08      14  1488.3    25.7 1484.75
    49.5 1484.59    73.5 1486.61    90.8 1483.68   117.9 1470.17   155.1 1459.27
   174.3 1455.56   183.9 1451.59   222.3 1447.98   255.9 1441.48   289.5 1428.99
   327.8 1426.91   337.2 1423.28   345.9 1421.22   360.3 1423.68     371  1426.6
   503.4 1427.81     519 1431.14   573.9  1432.3     583 1437.08   601.4 1442.95
   651.8 1468.98   673.4 1470.96   683.5  1479.4   689.3 1482.52   762.8 1513.68
#Mann= 10 ,-1 , 0
       0      .1       0     3.2     .05       0  217.96      .1       0
  325.34     .05       0   337.2    .045       0   360.3     .05       0
  449.76    .055       0  540.09     .05       0  647.47     .06       0
  754.85     .12       0
#XS Ineff= 2 , 0
                          373.99         1429.05
Permanent Ineff=
       F       F
Bank Sta=337.2,360.3
XS Rating Curve= 0 ,0
Exp/Cntr=0.3,0.1

Type RM Length L Ch R = 1 ,14691   ,368.5,377.9,383.6
XS GIS Cut Line= 2
     2475654.898       663669.32     2476338.235      664124.294
#Sta/Elev= 30
       0 1546.05   105.5 1532.24   153.6 1519.48   172.8 1512.63   197.2  1501.7
   260.7 1470.03   306.8 1444.95   327.6 1435.37     341 1432.07   374.6 1428.46
   384.3 1425.75   396.2 1420.28   413.1 1417.64   422.7 1420.01   446.7 1422.81
   488.6 1424.21   508.1 1423.13   581.3 1423.25   587.5 1424.08   601.9 1429.21
   621.3 1430.27   644.3 1444.69   676.1 1462.45   704.9 1481.88   710.7 1483.45
   730.3 1484.78   739.5 1493.46   746.2 1497.43   782.3    1513   820.9 1526.03
#Mann= 9 ,-1 , 0
       0     .05       0  128.12      .1       0  391.92     .05       0
   396.2    .045       0   422.7     .05       0  527.42    .035       0
  561.38     .05       0  662.92     .06       0  798.42      .1       0
#XS Ineff= 2 , 0
                          493.63         1430.74
Permanent Ineff=
       F       F
Bank Sta=396.2,422.7
XS Rating Curve= 0 ,0
Exp/Cntr=0.3,0.1

Type RM Length L Ch R = 1 ,14313   ,507.8,502.1,497.7
XS GIS Cut Line= 2
     2475497.581      663805.365     2475947.551      664496.617
#Sta/Elev= 30
       0 1547.63    33.7 1542.47    87.7 1531.56   155.2 1520.69     188 1512.29
   210.1 1505.42   250.6 1487.06   325.7    1443   350.2 1430.52   366.2 1424.69
   380.7 1422.03   398.1 1416.33   415.4 1413.51   421.1 1414.52     424 1415.98
   426.6 1417.29   431.4 1417.82   488.6 1416.41   522.1 1418.37     557 1422.05
   588.7 1427.56   610.7 1434.34   674.8 1457.73   684.2 1463.64   693.9    1471
   708.2 1472.66   727.6 1471.51   741.6 1477.27   788.3 1490.41   824.8 1502.49
#Mann= 6 ,-1 , 0
       0      .1       0  165.84      .1       0   398.1    .045       0
     424      .1       0  508.76      .1       0  657.02     .06       0
Bank Sta=398.1,424
XS Rating Curve= 0 ,0
Exp/Cntr=0.3,0.1

Type RM Length L Ch R = 1 ,13811   ,451.4,450,446.7
XS GIS Cut Line= 3
     2475093.021      664258.249     2475406.925      664523.183
2475718.17189161664789.093132477
#Sta/Elev= 30
       0 1533.21    44.1 1519.29   149.3 1479.42   166.3 1474.76   195.9 1469.87
   222.1 1463.11   286.3 1442.61     311  1433.1   321.5 1431.57   363.4 1421.57
   376.4 1419.83   397.9 1410.42   410.3    1408   422.6 1410.18   427.5 1411.13
   459.6 1411.31   484.2 1414.07   515.4 1415.53   526.3 1417.51   564.3 1433.27
   586.3 1437.13   597.7 1444.62   619.7 1452.74   637.4 1463.16   662.8 1465.51
   671.4 1472.33   691.3 1479.83   726.2 1491.26   779.3 1505.88   820.1 1520.23
#Mann= 8 ,-1 , 0
       0      .1       0  233.27      .1       0  370.04     .05       0
   397.9    .045       0   422.6     .05       0  491.36      .1       0
  619.95     .06       0  748.53      .1       0
Bank Sta=397.9,422.6
XS Rating Curve= 0 ,0
Exp/Cntr=0.3,0.1

Type RM Length L Ch R = 1 ,13361   ,335.8,337.6,338.3
XS GIS Cut Line= 3
     2474782.462      664642.774        2475124.      664870.168
2475467.14110839665104.866771177
#Sta/Elev= 30
       0 1507.29      34 1499.34    52.2  1493.2    96.4  1473.6   118.6 1465.01
   178.1 1450.85   271.5 1425.55   285.9 1420.39   317.8 1412.32   329.2 1408.38
   355.9 1405.98   392.6 1406.68   399.2 1405.55   404.2 1403.59   409.9 1402.89
   418.5 1403.03   432.8 1405.08   439.9 1406.18   503.7 1405.98   517.9 1407.65
   530.8 1410.69   539.6  1414.5   562.5 1428.95     622  1453.6   636.6 1462.37
   660.8  1463.9   670.5 1471.65   675.3 1474.54   762.6 1511.55     826 1540.59
#Mann= 11 ,-1 , 0
       0      .1       0   17.93      .1       0   57.44      .1       0
  153.43      .1       0  288.93     .05       0  346.28      .1       0
   399.2    .045       0   432.8      .1       0  489.63     .05       0
  561.69     .06       0  698.78      .1       0
Bank Sta=399.2,432.8
XS Rating Curve= 0 ,0
Exp/Cntr=0.3,0.1

Type RM Length L Ch R = 1 ,13023   ,412.7,412.4,410.1
XS GIS Cut Line= 2
2474655.77750622664922.957446007     2475236.445      665358.308
#Sta/Elev= 30
       0 1517.91    68.7 1484.22   159.2 1444.14   179.9  1437.2   199.9 1432.63
   246.6  1424.6   259.9 1423.33   273.3 1420.23   283.7 1414.61   293.7 1406.68
   299.2 1401.38   302.1 1399.97   307.8 1398.42   313.3 1398.25   323.7 1398.78
   328.7 1400.05   343.7 1403.09   359.2 1400.34   373.7 1400.06   418.7 1403.07
     460 1403.83   493.6 1408.78     540 1425.08   593.4 1452.08   608.6 1462.51
   630.7 1464.76   643.6 1474.14   648.6 1476.63   702.1 1498.27   725.7 1509.01
#Mann= 8 ,-1 , 0
       0      .1       0  120.67      .1       0  263.82      .1       0
   302.1    .045       0   328.7      .1       0  406.97      .1       0
  550.12     .06       0  693.27      .1       0
#XS Ineff= 2 , 0
                          343.14         1405.88
Permanent Ineff=
       F       F
Bank Sta=302.1,328.7
XS Rating Curve= 0 ,0
Exp/Cntr=0.3,0.1

Type RM Length L Ch R = 1 ,12611   ,452.1,450,447
XS GIS Cut Line= 3
 2474457.1532774665302.617518267     2474702.894      665462.368
     2475042.959      665691.417
#Sta/Elev= 30
       0 1544.49    59.1 1510.38   130.7    1471     145 1463.73   198.7 1440.21
   230.9 1421.22   254.8  1410.9   270.2 1401.06   283.4 1395.04   292.9 1393.32
   304.9 1393.77   310.7 1395.36     317 1397.04   344.2 1396.27     394 1398.53
   431.7 1397.94   460.5 1401.75   471.4 1405.88   518.1 1429.49   538.9 1438.48
   558.5 1450.03   582.3 1451.26   591.9 1457.77   610.4 1466.46   635.3 1484.97
   659.4 1494.83   685.3 1496.01   688.4 1497.31     698 1504.77   703.1 1507.63
#Mann= 6 ,-1 , 0
       0      .1       0   283.4    .045       0   310.7      .1       0
  326.31      .1       0  468.22     .06       0  611.81      .1       0
#XS Ineff= 2 , 0
                          392.96         1406.31
Permanent Ineff=
       F       F
Bank Sta=283.4,310.7
XS Rating Curve= 0 ,0
Exp/Cntr=0.3,0.1

Type RM Length L Ch R = 1 ,12161   ,365.1,373.4,381.5
XS GIS Cut Line= 3
2474223.38415946665733.225944762     2474460.861      665837.082
     2474832.308      666008.535
#Sta/Elev= 30
       0 1543.62   125.9 1472.51   164.8 1451.34   195.8 1435.65   208.9 1427.84
   217.6 1421.78   230.7  1409.7   239.4 1400.83   246.8 1391.83   249.8 1389.31
   252.5 1388.08   261.3 1387.57   265.7 1387.73     271 1389.55   296.5 1392.96
   379.5 1393.45   397.1  1395.3   406.7 1397.81   427.8 1396.35   442.8 1397.24
   516.8 1429.89   530.8 1433.17   543.2 1439.22   566.4 1448.48   574.1 1449.83
   591.7 1449.37   596.1 1450.86   605.6 1458.95   611.6 1462.08   668.3 1475.41
#Mann= 6 ,-1 , 0
       0      .1       0   249.8    .045       0     271      .1       0
  400.92     .05       0  529.08     .06       0  648.86      .1       0
#XS Ineff= 2 , 0
                          301.11         1403.44
Permanent Ineff=
       F       F
Bank Sta=249.8,271
XS Rating Curve= 0 ,0
Exp/Cntr=0.3,0.1

Type RM Length L Ch R = 1 ,11787   ,385.8,376.6,365.2
XS GIS Cut Line= 2
2474040.60901224665871.248971338     2474472.235      666440.996
#Sta/Elev= 30
       0 1548.77      27 1535.19   121.2 1480.31   161.2 1459.96   170.2 1454.47
   182.4 1445.78   202.3 1430.15   208.9 1423.78   215.5  1416.4   232.5 1395.57
   235.4 1392.64   240.4 1389.22   249.7 1386.68   275.6 1386.68   289.6 1384.74
   295.6 1382.86   300.6 1382.65   309.6 1383.13   314.9 1385.21   321.5  1391.4
   328.1 1392.94   354.6 1392.95   438.1 1396.65   526.6 1396.82   546.7 1395.52
     613 1398.75   632.8 1400.72   679.2 1408.01   705.7  1412.6   714.8    1415
#Mann= 4 ,-1 , 0
       0      .1       0   289.6    .045       0   314.9      .1       0
  345.61     .05       0
Bank Sta=289.6,314.9
XS Rating Curve= 0 ,0
Exp/Cntr=0.3,0.1

Type RM Length L Ch R = 1 ,11411   ,353.8,355.5,353.9
XS GIS Cut Line= 3
2473659.49858077666257.909838458     2474042.341      666394.449
      2474424.98      666540.326
#Sta/Elev= 30
       0 1647.44    16.2 1639.69    45.9 1622.28    87.8 1595.21   186.1 1537.35
   203.7 1525.59     237 1501.19   283.7 1463.49   309.2 1437.38     322 1426.09
   347.6 1407.89   355.9 1404.09   368.7 1400.95   372.9 1397.61   385.7 1383.62
   391.5 1380.03   406.4 1377.81   415.5 1377.97   419.7 1379.31     424 1382.59
   428.3 1384.28   445.4 1383.25   616.7 1384.22   667.5 1385.28   685.1  1388.1
   702.3 1387.26   762.2 1387.61   789.5 1393.69   809.3 1400.06     816 1403.27
#Mann= 6 ,-1 , 0
       0     .12       0   164.1      .1       0   391.5    .045       0
   419.7      .1       0  556.94     .05       0  786.48     .06       0
#XS Ineff= 2 , 0
                          429.35         1391.24
Permanent Ineff=
       F       F
Bank Sta=391.5,419.7
XS Rating Curve= 0 ,0
Exp/Cntr=0.3,0.1

Type RM Length L Ch R = 1 ,11055   ,363.2,368.2,365.7
XS GIS Cut Line= 2
2473597.56212147666606.0711864492474269.81354237666851.122498122
#Sta/Elev= 30
       0  1560.5    22.5 1548.08    69.4 1523.62    94.9 1511.25     129 1495.94
   154.2 1482.85   179.4 1467.86   243.9 1431.62     261  1421.4   279.3 1409.03
   299.3 1394.33   319.8 1378.28   324.8 1376.51   329.1 1375.95   346.1 1375.79
   355.7 1374.59   371.7 1372.49   379.1 1373.01   382.5 1374.63   388.7 1377.19
   418.5 1376.82   460.2 1380.27   554.7 1382.96   597.5 1386.76   675.5 1391.43
   691.1 1393.86   697.4 1396.62   703.7  1400.7   706.7 1401.55   715.5 1401.99
#Mann= 5 ,-1 , 0
       0      .1       0   355.7    .045       0   382.5      .1       0
  463.55     .05       0  681.49     .06       0
#XS Ineff= 2 , 0
                          397.78         1383.22
Permanent Ineff=
       F       F
Bank Sta=355.7,382.5
XS Rating Curve= 0 ,0
Exp/Cntr=0.3,0.1

Type RM Length L Ch R = 1 ,10687   ,305.9,299.7,291.1
XS GIS Cut Line= 2
2473425.70190678666880.6818182862474109.96403437 667116.12395951
#Sta/Elev= 30
       0 1494.39    34.9 1485.82    78.1 1472.38   131.6 1452.12   175.7 1431.75
     182 1428.24   185.1 1425.77   204.2 1408.74   216.8 1396.53   229.2 1386.68
   233.8 1383.68   246.5 1377.69   254.3 1370.72   259.1 1368.05   263.8 1367.55
   267.6 1367.73   275.4 1370.13     293 1371.44   309.9 1370.95     348 1372.56
   415.7 1373.95   471.5 1376.75   534.4 1377.02   563.7 1378.66   613.1 1383.67
     654 1394.09   669.5 1396.51   673.7 1398.93   686.4 1403.09   723.6 1404.33
#Mann= 6 ,-1 , 0
       0      .1       0   254.3    .045       0   275.4      .1       0
  388.85     .05       0  597.88     .06       0  701.31    .055       0
#XS Ineff= 2 , 0
                          349.95         1377.85
Permanent Ineff=
       F       F
Bank Sta=254.3,275.4
XS Rating Curve= 0 ,0
Exp/Cntr=0.3,0.1

Type RM Length L Ch R = 1 ,10388   ,88.3,94.5,97.3
XS GIS Cut Line= 3
2473355.79125518667263.0465607352473536.89313747667278.715666204
     2474112.601      667194.064
#Sta/Elev= 30
       0  1387.2    39.1 1389.37    75.2 1389.35   111.4 1386.56   148.5 1380.73
   175.6 1381.06   191.7 1379.51   195.8 1378.91   207.9 1374.71     220 1373.24
   236.1 1369.17   317.1 1368.47   334.8 1366.69   345.4 1364.72   357.5 1366.56
   381.8 1368.54   438.4 1368.57   462.6 1371.23   507.1 1374.02   556.9 1380.53
   608.2 1389.53   652.6 1393.21   660.7 1395.44   669.7 1401.06   676.9 1403.58
     689 1404.38   713.3 1404.25     734 1410.65   748.2 1413.58   763.7 1415.54
#Mann= 8 ,-1 , 0
       0      .1       0   39.54     .05       0  157.17      .1       0
  257.24     .05       0   334.8    .045       0   357.5     .05       0
  555.22     .06       0  753.87      .1       0
#XS Ineff= 2 , 0
          313.31 1371.75  385.95         1371.37
Permanent Ineff=
       F       F
Bank Sta=334.8,357.5
XS Rating Curve= 0 ,0
Exp/Cntr=0.5,0.3

Type RM Length L Ch R = 1 ,10293   ,72.1,71.3,70.9
XS GIS Cut Line= 3
2473305.25801528667372.9943842552473532.49938665667325.047413231
2474119.80832612667388.859989515
#Sta/Elev= 30
       0 1373.86    42.4 1373.67    87.4 1371.41   121.2 1371.46   144.8 1368.92
   156.9 1370.19   177.3 1374.54   218.2 1374.46   250.6 1370.27     311 1367.88
   371.3 1367.24   406.5 1365.58   423.6 1364.12   427.6  1364.2   431.9 1365.43
   439.7 1367.46     496 1366.33   556.4 1371.41   569.8  1379.6   596.6 1393.94
   620.8 1409.87   624.8 1411.86   631.5 1412.62     653 1412.75     657 1415.46
     665 1422.82   693.2  1433.5   737.4 1447.51   769.4 1456.17     823 1468.18
#Mann= 7 ,-1 , 0
       0     .05       0  220.12      .1       0  303.85     .05       0
   406.5    .045       0   431.9     .05       0  631.76     .06       0
  734.78      .1       0
#XS Ineff= 2 , 0
          380.94 1366.13  443.99         1365.95
Permanent Ineff=
       F       F
Bank Sta=406.5,431.9
XS Rating Curve= 0 ,0
Exp/Cntr=0.5,0.3

Type RM Length L Ch R = 1 ,10222   ,69.5,69.4,69.3
XS GIS Cut Line= 3
2473314.91457758 667425.367287952473557.03901323667407.801625365
2474127.56813178667437.079341102
#Sta/Elev= 30
       0    1373   180.3 1369.96   216.4 1368.37   256.5 1368.62   308.6 1362.95
   321.5 1362.59   334.2 1362.83   351.1 1366.65   360.6 1367.04   373.1 1365.76
   388.3 1362.23   396.7 1360.58   412.7 1360.87   424.7  1362.3   436.7 1366.35
   452.7  1366.4   472.8  1368.2   488.8  1367.3   492.8 1368.99   512.8 1382.91
   552.9 1403.15   568.9 1413.97   576.9 1415.86   600.9 1415.18   604.9 1417.21
     617 1427.81     677 1449.77   737.1 1468.52   792.1 1482.88     814 1487.28
#Mann= 5 ,-1 , 0
       0     .05       0   388.3    .045       0   424.7     .05       0
  523.91     .06       0  727.09      .1       0
#XS Ineff= 2 , 0
          358.06 1372.05   473.2         1373.19
Permanent Ineff=
       F       F
Bank Sta=388.3,424.7
XS Rating Curve= 0 ,0
Exp/Cntr=0.5,0.3

Type RM Length L Ch R = 1 ,10152   ,238.1,241.5,243.7
XS GIS Cut Line= 2
2473287.78782161667472.478394906     2474132.498      667496.438
#Sta/Elev= 30
       0 1372.99     227 1367.94   255.1  1366.4   311.1 1365.93   355.1 1366.76
   391.1 1361.28   416.5 1360.41   431.1 1358.43   439.1 1360.48   447.1 1363.22
   463.1 1365.42   467.1 1365.78   476.1 1364.02   483.2 1365.86   487.2 1369.49
   495.5 1381.06     503 1386.95   523.2 1397.82   543.2 1406.11   559.2 1416.62
   567.2 1418.06   591.2  1416.9   599.2 1422.03   607.2 1429.55   611.2  1432.3
   627.2  1437.7   695.2 1464.38   778.9 1494.65   814.6 1504.98     845  1511.7
#Mann= 5 ,-1 , 0
       0     .05       0   416.5    .045       0   439.1     .05       0
  560.98     .06       0   662.1      .1       0
#XS Ineff= 2 , 0
          353.71 1371.52  467.99         1371.36
Permanent Ineff=
       F       F
Bank Sta=416.5,439.1
XS Rating Curve= 0 ,0
Exp/Cntr=0.3,0.1

Type RM Length L Ch R = 1 ,9911    ,428.5,427.4,421.1
XS GIS Cut Line= 3
2473315.36604817667654.777132477      2473730.32      667724.032
     2474131.799      667803.668
#Sta/Elev= 30
       0 1380.38    20.4 1380.28      48 1378.53     142 1368.34     194 1366.04
   368.4 1362.52   404.9 1358.52     413 1356.16   421.1 1355.48   425.2 1356.03
   429.3 1358.72   437.4 1372.09   441.5 1377.01   450.7 1386.35   478.2  1411.7
   482.3 1414.43   486.4 1415.39   502.7 1415.05   508.6 1416.32   510.8 1417.65
   514.3  1421.8   519.3 1430.57   523.1 1436.06   527.2 1439.25   567.9 1462.58
   610.6 1488.92   657.6 1513.27   699.1 1532.25     780 1563.46     830 1578.65
#Mann= 5 ,-1 , 0
       0     .05       0   404.9    .045       0   429.3     .05       0
  479.49     .06       0  585.47      .1       0
#XS Ineff= 2 , 0
          368.12 1369.76
Permanent Ineff=
       F       F
Bank Sta=404.9,429.3
XS Rating Curve= 0 ,0
Exp/Cntr=0.3,0.1

Type RM Length L Ch R = 1 ,9483    ,307.1,322.6,342.8
XS GIS Cut Line= 3
     2473240.856      668005.5712473452.78039703668130.211228823
     2474048.307      668155.793
#Sta/Elev= 30
       0 1369.84    62.5 1365.85   177.7 1361.71   251.8 1356.73   363.9    1357
   379.9 1357.67     402 1355.62     416 1355.98     420 1354.93     428 1351.59
     436 1351.18     460 1354.98     464  1355.9     476 1356.42     480 1358.03
   505.6 1377.11   528.1 1391.61     540 1401.18   544.1 1403.59   569.3 1405.93
   592.1 1405.29   596.1  1405.9   600.2  1408.8   608.2 1420.39   613.1 1422.93
   624.6 1425.76   689.9 1437.87   739.8 1448.79   778.2 1458.28   841.9 1476.75
#Mann= 5 ,-1 , 0
       0     .05       0     420    .045       0     460      .1       0
  546.83     .06       0  648.24      .1       0
#XS Ineff= 2 , 0
          378.46 1362.05
Permanent Ineff=
       F       F
Bank Sta=420,460
XS Rating Curve= 0 ,0
Exp/Cntr=0.3,0.1

Type RM Length L Ch R = 1 ,9161    ,319.6,324.2,329.3
XS GIS Cut Line= 3
     2473195.242      668072.521     2473484.337      668386.627
     2473771.676      668679.222
#Sta/Elev= 30
       0 1366.61   139.1 1359.93   216.5 1354.46   258.7 1353.92   296.8 1352.96
   351.1 1355.54   369.3 1352.79   400.9 1352.39   414.6 1350.52   427.3 1348.48
   438.5 1348.91   444.1 1350.86   494.5 1389.77   510.3 1404.05   522.6    1417
   527.8 1420.41   533.4 1421.87   561.8 1422.72   567.4 1424.22     573 1429.83
   581.5 1449.45   584.2 1454.43   589.8  1459.2   629.1 1482.97   670.1 1503.45
   690.8 1509.15   707.6 1511.41   738.6 1509.53   791.7 1503.12     837 1500.55
#Mann= 7 ,-1 , 0
       0     .05       0   258.7      .1       0   414.6    .045       0
   444.1      .1       0  488.28     .06       0  610.46      .1       0
  782.45      .1       0
#XS Ineff= 2 , 0
          351.62 1365.31
Permanent Ineff=
       F       F
Bank Sta=414.6,444.1
XS Rating Curve= 0 ,0
Exp/Cntr=0.3,0.1

Type RM Length L Ch R = 1 ,8837    ,421,425.8,427.6
XS GIS Cut Line= 2
     2472999.828      668166.556     2473401.391      668885.027
#Sta/Elev= 30
       0 1369.24    71.6 1361.68   229.5 1353.79     264  1350.1   302.2 1349.25
   385.3 1349.83   389.9    1349   396.3 1345.07   399.5 1343.27     408 1342.22
   417.4 1342.74   424.1 1344.87   434.5 1348.96   443.3 1354.65   502.3 1404.43
   530.7 1426.16   541.1 1429.87     564 1429.23   569.7 1430.03   573.2 1432.39
   575.6 1435.75   582.3 1447.85   587.3 1455.19   591.5 1459.11     602  1466.1
   651.1  1495.2   684.3 1517.21     699 1525.85     749  1554.2   823.1 1593.78
#Mann= 7 ,-1 , 0
       0    .055       0  153.48     .05       0   364.5      .1       0
   396.3    .045       0   424.1      .1       0  468.54     .06       0
  572.59      .1       0
#XS Ineff= 2 , 0
          380.47 1359.22
Permanent Ineff=
       F       F
Bank Sta=396.3,424.1
XS Rating Curve= 0 ,0
Exp/Cntr=0.3,0.1

Type RM Length L Ch R = 1 ,8411    ,302.9,300,297.1
XS GIS Cut Line= 3
     2472691.302       668366.16     2472842.259      668751.525
     2472989.545      669132.787
#Sta/Elev= 30
       0 1374.28   112.5 1359.95   185.3 1354.13   234.7 1352.03   249.9 1344.79
   268.7 1340.01   288.6  1340.4   305.7 1343.59   327.5  1342.5   364.4 1344.32
   374.5 1344.24   391.7 1339.52   410.7 1337.41   417.5  1337.6   426.1 1340.39
   426.1 1340.44   430.3 1343.89   438.9 1354.01   447.5 1368.97   468.9 1375.83
   500.4 1392.71   525.1  1409.5   533.3 1411.12   558.7 1411.01   563.3 1412.34
   571.9 1419.49   584.7 1435.56     589 1438.43   692.1 1496.71   822.6 1566.45
#Mann= 6 ,-1 , 0
       0    .055       0  196.51      .1       0   391.7    .045       0
   426.1      .1       0  496.22     .06       0  596.04      .1       0
#XS Ineff= 2 , 0
          363.08 1350.52
Permanent Ineff=
       F       F
Bank Sta=391.7,426.1
XS Rating Curve= 0 ,0
Exp/Cntr=0.3,0.1

Type RM Length L Ch R = 1 ,8111    ,443.3,450,451.1
XS GIS Cut Line= 3
     2472343.018      668496.906     2472563.511      668846.271
     2472771.444      669201.748
#Sta/Elev= 30
       0 1374.06    30.7 1369.06      78 1363.28   182.1    1353   191.5 1349.17
   201.8  1343.1     210 1341.06   381.7 1339.33   395.6 1335.35   404.3 1333.35
     413 1333.07   424.7 1335.19   433.5 1336.98   450.9 1337.86   465.6 1336.57
   469.5 1337.04   474.1 1339.17   486.1 1353.97   492.6 1360.48   512.4 1374.37
     539 1391.46   562.1 1410.75   570.1 1413.42   585.5 1413.48   589.9 1414.59
   594.6 1418.42   603.8 1429.92   613.1 1436.56   775.3 1539.82     825 1568.55
#Mann= 7 ,-1 , 0
       0     .05       0  126.48    .055       0  339.09     .05       0
   395.6    .045       0   424.7      .1       0  549.78     .06       0
  654.61      .1       0
#XS Ineff= 2 , 0
          380.94 1345.83
Permanent Ineff=
       F       F
Bank Sta=395.6,424.7
XS Rating Curve= 0 ,0
Exp/Cntr=0.3,0.1

Type RM Length L Ch R = 1 ,7661    ,305,308.3,309.4
XS GIS Cut Line= 3
     2472008.679      668582.579     2472141.699      668969.903
     2472269.363      669359.006
#Sta/Elev= 30
       0 1377.33    18.7  1369.3    34.2 1368.92    89.1 1359.48   101.8 1359.13
   178.2 1348.52   232.9 1337.09   313.3 1335.72   347.1 1332.88   389.4 1332.24
   393.7 1331.14   397.9 1328.78   406.3 1328.19   423.2 1329.34   431.6 1331.29
   528.4 1334.06   549.5 1329.96   562.1 1331.19   566.5 1333.75   579.1 1347.48
   587.4 1354.17   612.6 1370.84   642.1 1386.84   658.9  1398.9   667.4 1400.72
   684.2 1400.22   688.4 1402.21   696.8 1410.97   703.9 1415.07     819    1461
#Mann= 7 ,-1 , 0
       0      .1       0   29.31     .05       0   393.7    .045       0
   431.6     .05       0  480.18      .1       0  579.02     .06       0
  677.87      .1       0
#XS Ineff= 2 , 0
           373.7 1337.13
Permanent Ineff=
       F       F
Bank Sta=393.7,431.6
XS Rating Curve= 0 ,0
Exp/Cntr=0.3,0.1

Type RM Length L Ch R = 1 ,7353    ,85.2,87.4,88.6
XS GIS Cut Line= 2
2471769.52136904668716.3174106932471926.60052735669399.393113367
#Sta/Elev= 30
       0 1364.77    31.4 1349.88    43.7 1347.85    60.1 1339.36    76.5 1336.22
   158.6 1331.88   306.4 1329.03   322.8 1329.56     331 1328.04   339.2 1325.94
   351.5 1325.42   356.9 1326.12   363.8 1328.59   367.9 1329.35   384.3 1328.72
     409 1329.48   429.5 1328.09   445.9  1328.3     450 1330.04   458.2 1337.28
   462.3 1338.57   478.8 1339.59   524.1 1345.85   564.9 1348.72   597.8 1353.95
   630.5  1360.5   650.6 1362.36   659.3 1365.17   679.9 1374.41   700.9 1374.71
#Mann= 8 ,-1 , 0
       0     .05       0   85.01      .1       0   182.8     .05       0
     331    .045       0   363.8     .05       0  378.39      .1       0
  573.97     .05       0  671.76     .06       0
#XS Ineff= 2 , 0
          292.89 1336.86
Permanent Ineff=
       F       F
Bank Sta=331,363.8
XS Rating Curve= 0 ,0
Exp/Cntr(USF)=0,0
Exp/Cntr=0.5,0.3

Type RM Length L Ch R = 1 ,7265    ,66.3,64.8,62.7
XS GIS Cut Line= 2
2471701.03067443668710.4525864822471828.45724038669443.032277327
#Sta/Elev= 30
       0 1378.14    32.9 1368.47    49.2 1362.61    57.3 1358.65    60.7 1355.78
    65.4 1350.28    69.5 1347.21    85.7 1344.78    93.8 1341.19   109.1 1341.08
   118.2 1338.07   122.2 1337.67   150.7 1336.31   227.8 1330.61   280.6 1328.75
   325.2 1328.41   353.7 1326.89   365.9 1325.57   394.3 1326.68   471.4 1328.94
   516.1 1328.99   548.6  1327.5     577 1327.61   609.5 1329.48   621.6  1331.2
   637.9 1334.81   686.6 1351.69   706.9 1356.73   727.2 1360.33   743.6 1366.42
#Mann= 7 ,-1 , 0
       0      .1       0    3.56     .05       0  101.12      .1       0
  296.22     .05       0   353.7    .045       0   394.3     .05       0
  686.44     .06       0
#XS Ineff= 4 ,-1
       0   325.2  1333.8   325.2     353  1326.8     395     516  1326.8
     516     700  1333.8
Permanent Ineff=
       F       F       F       F
Bank Sta=353.7,394.3
XS Rating Curve= 0 ,0
Exp/Cntr(USF)=0,0
Exp/Cntr=0.5,0.3

Type RM Length L Ch R = 1 ,7200    ,73.8,73.3,73
XS GIS Cut Line= 2
  2471618.442474668722.8976942172471788.20750717669467.989741825
#Sta/Elev= 30
       0 1354.81    12.3 1354.45    20.5 1353.41      41 1352.05    77.9 1351.78
    86.1 1349.82    97.1 1344.87   109.4 1341.35   123.1 1339.76   147.7 1338.75
     160 1336.69   184.6 1334.52   209.2 1333.54   257.5 1329.09   280.9 1329.15
     320 1327.74   344.4 1327.55   371.1 1325.78   385.6 1324.32   401.2 1325.67
   430.8 1328.03   475.9 1329.24     599 1326.66   631.8 1327.97   648.2 1330.94
   672.8 1338.15   701.5 1344.75   746.7 1352.59   755.4 1355.54   764.2 1360.53
#Mann= 5 ,-1 , 0
       0      .1       0  297.28     .05       0   371.1    .045       0
   401.2     .05       0  688.39     .06       0
#XS Ineff= 2 , 0
          306.23 1333.75  479.02         1333.29
Permanent Ineff=
       F       F
Bank Sta=371.1,401.2
XS Rating Curve= 0 ,0
Exp/Cntr=0.5,0.3

Type RM Length L Ch R = 1 ,7127    ,156.3,141,106.6
XS GIS Cut Line= 3
2471553.16161648668790.3971085792471666.88099522669253.265670554
2471777.25531727669462.575317528
#Sta/Elev= 30
       0  1378.7    29.3 1372.24    45.8 1366.91    99.4 1345.19   111.7 1339.26
     124 1335.36   136.4 1332.61   150.5 1331.03   185.9 1329.15   255.9  1327.6
   309.4  1325.1   329.1 1324.98   338.3 1323.21   342.3 1323.06   358.8 1324.94
   375.3 1327.09   428.9 1329.28   437.1 1328.67   453.6 1328.79   470.1 1327.21
   510.1    1326   536.4 1326.62   579.2 1326.42   600.6  1327.8   605.1 1328.63
   618.7 1334.08   627.7 1336.56   673.6  1343.8   693.9 1348.34   713.3 1353.68
#Mann= 5 ,-1 , 0
       0      .1       0  240.78     .05       0   329.1    .045       0
   358.8     .05       0  641.04     .06       0
#XS Ineff= 2 , 0
                          426.34         1335.52
Permanent Ineff=
       F       F
Bank Sta=329.1,358.8
XS Rating Curve= 0 ,0
Exp/Cntr(USF)=0,0
Exp/Cntr=0.5,0.3

Type RM Length L Ch R = 1 ,6986    ,78.5,79.9,90.5
XS GIS Cut Line= 4
2471373.25377876668916.2150081642471429.93062698669092.360067583
2471569.97653204  669168.2035678 2471765.0530698669469.108245406
#Sta/Elev= 30
       0 1386.88    54.2 1371.24    95.3 1357.98   124.1 1346.19   145.7 1338.92
   158.3 1333.02   169.1 1329.29     175 1328.24     185 1328.71   199.3 1328.04
   217.8 1325.33   243.6 1323.26   249.6  1322.2   257.6 1321.84     276 1321.98
   290.6  1323.1   313.3 1324.12   333.1 1325.99   385.6 1327.37   430.7 1327.44
   490.5 1325.18   526.1 1326.38   552.5 1325.92   576.3 1327.48   585.9 1329.09
   604.9 1336.17   609.7 1337.32   661.9 1343.37     684 1348.24   702.9 1354.48
#Mann= 4 ,-1 , 0
       0      .1       0   243.6    .045       0   290.6     .05       0
  678.23     .06       0
#XS Ineff= 2 , 0
          192.45    1330  342.05         1329.69
Permanent Ineff=
       F       F
Bank Sta=243.6,290.6
XS Rating Curve= 0 ,0
Exp/Cntr(USF)=0,0
Exp/Cntr=0.5,0.3

Type RM Length L Ch R = 1 ,6906    ,61.4,68.1,78.5
XS GIS Cut Line= 4
2471337.02757298668928.2191459592471394.41940673669149.036915808
2471530.23218619669206.3016981422471727.73820717669492.334642497
#Sta/Elev= 30
       0 1384.08    64.8 1368.29   118.5  1356.8   168.1 1341.63   184.6 1331.53
   188.7 1331.19   197.1  1333.6   205.3 1333.56   217.7 1336.88   228.2 1332.57
   235.9 1327.19   248.1 1323.05   253.5 1320.73   258.9 1320.11   277.8 1321.69
   293.6 1322.97   306.2 1322.78   318.4  1325.1   328.4  1325.5   350.1 1324.78
   382.1 1325.64   405.4 1325.09     420 1325.95   517.2 1323.94   551.7 1327.02
   614.4 1337.54   643.6 1340.37   701.9 1344.09   714.4 1345.85   723.1 1348.42
#Mann= 4 ,-1 , 0
       0      .1       0   248.1    .045       0   277.8      .1       0
  353.32     .05       0
#XS Ineff= 1 ,-1
     431     600    1328
Permanent Ineff=
       F
Bank Sta=248.1,277.8
XS Rating Curve= 0 ,0
Exp/Cntr=0.5,0.3

Type RM Length L Ch R = 1 ,6838    ,263,259.5,253.8
XS GIS Cut Line= 2
2471199.84839731669038.0816249182471675.67984453669496.170204615
#Sta/Elev= 30
       0 1368.64    24.2 1364.12    81.8 1356.35   120.6 1354.15   162.7 1348.82
   192.2 1346.66   208.8 1343.04   226.1 1337.72   237.2 1330.55   243.4 1322.93
   248.3 1320.18   254.4 1320.08   268.5 1322.06   288.3 1322.84   302.5 1321.93
   324.1 1324.39   359.1 1324.68   384.5 1324.69   424.1 1322.97   445.3 1323.25
     476 1325.54   497.7 1328.33     601 1338.05     608 1338.03   618.3 1335.26
   624.1 1334.93   629.8 1337.84   641.4 1345.89   653.7 1349.92   660.5 1351.06
#Mann= 4 ,-1 , 0
       0      .1       0   243.4    .045       0   268.5      .1       0
   307.1     .05       0
Bank Sta=243.4,268.5
XS Rating Curve= 0 ,0
Exp/Cntr(USF)=0,0
Exp/Cntr=0.3,0.1

Type RM Length L Ch R = 1 ,6579    ,308.6,301.5,289.7
XS GIS Cut Line= 2
2471018.93882204669272.0127876732471561.09587241669640.984607347
#Sta/Elev= 30
       0 1392.02    33.6    1388    53.8 1384.35    82.5 1376.86    86.9 1375.02
    96.9 1368.77   111.1 1368.12   115.9 1366.81   125.6 1361.06   148.8 1352.43
   169.1  1342.4   182.9 1334.77   206.3 1319.74   212.1 1317.26   217.9 1317.04
   227.2 1317.23   243.8 1319.75   261.1 1319.63   324.4 1321.66   493.3 1321.32
   522.3 1322.05   537.4 1323.86   546.5 1323.76   552.5    1325     572 1335.89
   585.2 1341.19   620.9 1351.23   635.3 1354.58     645 1355.82   655.8 1358.75
#Mann= 6 ,-1 , 0
       0      .1       0   206.3    .045       0   243.8      .1       0
  345.76     .05       0  546.92      .1       0  631.45     .06       0
#XS Ineff= 2 , 0
                          489.79         1328.73
Permanent Ineff=
       F       F
Bank Sta=206.3,243.8
XS Rating Curve= 0 ,0
Exp/Cntr=0.3,0.1

Type RM Length L Ch R = 1 ,6277    ,325.5,324.5,323.6
XS GIS Cut Line= 2
2470826.16439339669628.0472676982471492.05586629669702.794925143
#Sta/Elev= 30
       0 1356.29    36.8 1346.19      73 1334.99   101.2 1330.33   109.3 1330.25
   125.4 1332.31   137.4 1332.86   201.8 1331.58   205.9 1329.99   217.9  1318.2
     222 1315.71     226 1314.53     234 1314.09   249.2 1315.57   258.2 1316.36
   278.3 1314.67   290.4 1317.41   298.4 1317.82     395 1316.74   467.5 1318.66
     548 1318.37   564.1 1318.88   576.2  1320.4   592.3 1319.95   596.3 1320.78
   600.5 1322.85   620.5 1335.08   632.5 1341.33   644.6  1344.7   670.1 1353.69
#Mann= 7 ,-1 , 0
       0     .05       0   43.41      .1       0  153.43     .05       0
     222    .045       0   249.2     .05       0  462.79      .1       0
  669.03     .06       0
#XS Ineff= 2 , 0
                          476.07         1322.35
Permanent Ineff=
       F       F
Bank Sta=222,249.2
XS Rating Curve= 0 ,0
Exp/Cntr=0.3,0.1

Type RM Length L Ch R = 1 ,5953    ,221.1,235.4,254.6
XS GIS Cut Line= 3
2470862.18255698669704.6662429392470956.66879518669920.290850286
2471402.77400988669923.116111591
#Sta/Elev= 30
       0 1343.05    19.9 1336.69    29.4 1331.33    53.7 1324.19    72.3 1326.29
   153.9 1321.23   169.1 1321.48   193.4 1318.98   232.9 1317.74   249.5 1313.52
   257.5 1312.81   329.5 1312.61   393.5 1314.71   421.5 1313.59   437.5 1314.14
   449.5 1311.65   465.5 1312.54   474.6 1311.41   485.5 1309.62   506.4 1311.45
   525.5 1310.83   529.5 1312.54   537.5 1320.18   565.5 1341.42   585.1 1352.77
   605.2 1361.79     646 1376.23   665.5  1386.7   673.3 1388.56   681.5  1388.7
#Mann= 5 ,-1 , 0
       0      .1       0    29.4     .05       0   474.6    .045       0
   506.4      .1       0   605.2     .06       0
Bank Sta=474.6,506.4
XS Rating Curve= 0 ,0
Exp/Cntr=0.3,0.1
